HEC-RAS study SndlckCrk.prj: SndlckCrk

--- SndlckCrk.g01 (geometry) --- (continued)

Type RM Length L Ch R = 1 ,28696.7 ,135.1,138.6,142.2
XS GIS Cut Line= 3
      1866172.37      301426.804      1866260.33      302777.974
      1866274.99      302902.585
#Sta/Elev= 30
       0 1929.18    19.9 1926.85    79.6 1916.57    99.6 1914.22   119.5 1909.08
   129.4 1905.77   139.4  1901.2   169.2 1881.88   179.2 1879.52   189.2 1874.39
     239 1838.29   268.8 1814.61   278.8 1811.36   288.7 1806.44   358.4 1748.94
   378.3 1741.08   398.2 1725.93   408.2 1719.78   418.2 1716.14   423.9 1715.47
   438.1 1714.92   438.9 1714.93   836.3 1719.93  1055.4 1720.31    1135 1722.09
  1224.6 1725.65  1392.6 1734.15  1431.2 1735.07  1450.6 1737.13  1479.5 1743.87
#Mann= 3 , 0 , 0
       0     .06       0   423.9    .045       0   438.9     .06       0
Bank Sta=423.9,438.9
XS Rating Curve= 0 ,0
Exp/Cntr=0.3,0.1

Type RM Length L Ch R = 1 ,28558   ,270.5,262.9,251.3
XS GIS Cut Line= 3
     1866072.193      301297.714     1866072.193      301662.587
     1866075.451       303047.15
#Sta/Elev= 30
       0 1983.53    19.7 1979.59    78.9 1975.04   167.6 1970.76   187.4 1966.14
   207.1 1957.09     217  1954.9   226.8 1950.88   295.8 1900.69   315.6 1893.72
   335.3 1880.04   364.9 1861.13   384.8 1847.11   394.8 1842.26   404.7 1839.54
   484.4 1775.72   494.4 1770.42   504.3 1768.14   554.1 1731.38   564.1 1724.91
     574  1720.4   603.7  1715.7   618.7 1714.79   623.9 1714.77  1032.2 1720.35
  1201.6  1721.4    1341  1724.9  1639.9 1734.75  1719.6 1743.43  1749.4  1750.4
#Mann= 3 , 0 , 0
       0     .06       0   603.7    .045       0   618.7     .06       0
Bank Sta=603.7,618.7
XS Rating Curve= 0 ,0
Exp/Cntr=0.3,0.1

Type RM Length L Ch R = 1 ,28293.6 ,69.5,73.2,80.8
XS GIS Cut Line= 3
     1865840.489      301390.631     1865837.695      301942.562
     1865993.864      303005.999
#Sta/Elev= 30
       0 1956.21     9.9 1953.66    19.7 1953.03    39.4 1946.13    59.1 1941.81
   108.4 1936.48   177.4 1931.67   187.3 1928.99   197.1  1923.1     207 1922.43
   216.8 1916.35   295.7 1857.62   305.5 1855.79   315.4  1850.9   384.4 1803.32
   404.1 1796.66   473.1  1744.4   492.8  1737.6   512.5  1725.7   522.4 1721.76
   542.1 1715.78   556.3 1714.61   561.9 1714.58   571.3  1714.6   691.3 1714.71
  1387.9 1725.42  1487.4 1729.66  1567.1 1735.85  1596.9 1740.96  1626.8 1752.39
#Mann= 3 , 0 , 0
       0     .06       0   556.3    .045       0   571.3     .06       0
Bank Sta=556.3,571.3
XS Rating Curve= 0 ,0
Exp/Cntr=0.3,0.1

Type RM Length L Ch R = 1 ,28221.9 ,1022.6,1025.8,1029.3
XS GIS Cut Line= 3
     1865730.124      301245.589     1865746.413      301587.658
     1865863.694      303096.017
#Sta/Elev= 30
       0 1962.68    19.6 1963.51    78.3 1953.69    97.8 1946.81   146.8 1923.89
   166.3 1919.42   195.7 1906.64   215.3 1900.32   244.6 1895.82   372.3 1888.79
   382.3  1886.2     432 1852.89     442  1851.6   451.9 1846.19   531.6 1794.04
   541.5 1792.29   551.5 1787.76   621.2 1739.85   641.1 1732.77   670.9 1716.16
   680.9 1714.56   681.8 1714.56   696.8  1714.6     870 1714.69  1487.1 1720.93
  1586.6 1724.22  1706.1 1734.84  1745.9 1745.51  1825.5 1758.15  1855.4 1765.88
#Mann= 3 , 0 , 0
       0     .06       0   681.8    .045       0   696.8     .06       0
Bank Sta=681.8,696.8
XS Rating Curve= 0 ,0
Exp/Cntr=0.3,0.1

Type RM Length L Ch R = 1 ,27195.9 ,458.3,458.4,454.9
XS GIS Cut Line= 3
     1864892.871       301141.34     1865195.846      302933.127
     1865225.166      303102.532
#Sta/Elev= 30
       0 1861.66   169.7 1848.62   349.5 1840.01   389.4 1835.17   419.4 1828.32
   439.3 1824.83   479.3 1814.28   499.2 1808.01   519.2 1799.58   539.2  1794.2
   609.1 1763.05     619 1759.45     629 1757.73   698.9 1724.28   708.9 1720.08
   718.9 1717.42   738.9 1716.39   847.5 1714.83   862.5 1714.62   868.7  1714.6
   978.5 1714.65  1068.4  1716.6  1158.2  1717.4  1347.9 1717.94  1587.6 1721.78
  1697.4 1725.22  1787.3 1729.51    1865 1736.48  1960.5 1741.78  1989.2  1742.6
#Mann= 3 , 0 , 0
       0     .06       0   847.5    .045       0   862.5     .06       0
Bank Sta=847.5,862.5
XS Rating Curve= 0 ,0
Exp/Cntr=0.3,0.1

Type RM Length L Ch R = 1 ,26736.8 ,713.6,721.2,727.7
XS GIS Cut Line= 3
     1864629.472      301596.701     1864879.248      303059.931
     1864862.959      303222.821
#Sta/Elev= 30
       0 1945.33    19.9  1939.1    49.8 1926.81    69.7 1922.63   129.5 1901.84
   139.5 1898.73   159.4  1895.4   219.2 1871.82   249.1 1858.76     259 1856.37
   308.8 1825.62   338.7 1813.92   348.7 1812.73   358.6 1806.82   368.6 1799.93
   388.5 1783.25   438.3 1736.31   448.3  1735.4   458.3  1729.9   498.1 1717.43
   593.5 1712.98   597.7 1712.97   608.5 1713.49   647.6 1715.04   826.9 1716.34
   996.2 1721.31    1325 1727.71  1503.6 1736.59  1619.2 1758.37  1648.1 1760.68
#Mann= 3 , 0 , 0
       0     .06       0   593.5    .045       0   608.5     .06       0
Bank Sta=593.5,608.5
XS Rating Curve= 0 ,0
Exp/Cntr=0.3,0.1

Type RM Length L Ch R = 1 ,26015.1 ,881.1,883.1,885.2
XS GIS Cut Line= 2
     1864587.694      301522.471     1864179.414      303180.719
#Sta/Elev= 30
       0 1937.84    79.9 1926.31   139.8 1920.53   239.7 1898.33   279.6 1886.72
   289.6 1882.83   309.6 1872.39   329.6 1865.54   369.5 1837.69   399.5 1819.05
   409.5 1813.57   419.4 1812.63   479.4 1771.84   509.3 1749.49   519.3 1747.25
   529.3 1741.37   549.3 1726.46   559.3 1720.49   569.3 1717.26   601.5 1712.16
   616.5 1711.49   709.1  1711.1   808.9 1712.13  1048.6 1717.89  1288.3 1717.74
  1388.2 1721.64    1548 1730.99  1577.9 1731.85  1657.8 1739.43  1707.8 1741.15
#Mann= 3 , 0 , 0
       0     .06       0   601.5    .045       0   616.5     .06       0
Bank Sta=601.5,616.5
XS Rating Curve= 0 ,0
Exp/Cntr=0.3,0.1

Type RM Length L Ch R = 1 ,25131.6 ,405.6,406.9,408.8
XS GIS Cut Line= 3
     1864117.516      301271.651     1864055.618      301506.213
     1863645.135       303017.83
#Sta/Elev= 30
       0 1888.34     9.7 1887.85    48.5 1880.56    77.6 1877.07      97 1876.67
     165 1857.54   174.7 1855.84   184.4 1856.61   203.8 1851.36   262.5 1843.48
   282.5 1842.95   322.4 1834.36   362.3 1821.43   382.3 1819.04   432.2 1782.95
   462.1 1759.32   472.1 1758.91     502 1736.86   531.9 1717.02   541.9 1712.06
     553  1710.3   561.8 1710.15     568 1710.21   821.2 1713.87  1170.4  1714.2
  1439.8 1719.36  1659.3 1728.27  1719.2 1738.97  1729.1 1739.55    1809    1756
#Mann= 3 , 0 , 0
       0     .06       0     553    .045       0     568     .06       0
Bank Sta=553,568
XS Rating Curve= 0 ,0
Exp/Cntr=0.3,0.1

Type RM Length L Ch R = 1 ,24724.1 ,1253.5,1254.6,1250.3
XS GIS Cut Line= 3
     1863798.077      301294.307     1863579.396      301920.391
     1863069.222      303234.169
#Sta/Elev= 30
       0 1938.48    39.6 1918.72    59.4 1914.32   138.6  1873.5   158.4    1869
   217.8 1838.39   237.6 1831.17   247.4 1831.33   257.4 1828.14   336.5 1791.97
   356.3 1787.41   376.1 1774.16     386 1760.18   415.7 1730.12   435.5 1720.51
   534.5 1713.61   633.5  1709.7   647.7  1709.7   662.7  1709.7    1053  1713.8
  1262.9  1719.9  1362.9 1728.94  1392.8 1738.04  1432.8 1754.43  1462.8 1757.63
  1642.7 1750.59  1732.7 1726.47  1752.7 1724.93  1892.6 1723.33  2072.5 1725.05
#Mann= 3 , 0 , 0
       0     .06       0   647.7    .045       0   662.7     .06       0
Bank Sta=647.7,662.7
XS Rating Curve= 0 ,0
Exp/Cntr=0.3,0.1

Type RM Length L Ch R = 1 ,23466.8 ,303.7,278.7,254.9
XS GIS Cut Line= 3
      1863322.24      301046.797       1862872.7      301301.022
     1862456.515      303178.016
#Sta/Elev= 30
       0 1925.34    29.8 1915.78    79.4 1887.44   109.2 1881.77   168.8 1862.09
   188.7 1861.58   327.7 1837.68   427.1 1829.08   466.8  1820.5   536.4 1797.47
   616.1 1756.53     626 1756.23   685.8 1725.82   759.2 1709.71   765.5  1709.7
   774.2 1709.76  1024.5  1721.1    1154 1744.39  1363.2 1759.94  1482.7 1774.78
  1642.1 1775.01  1711.8 1762.67  1781.6 1764.97  1861.3 1758.41  1960.9 1771.24
  2030.6 1770.92    2180 1757.74  2349.4 1761.28  2399.2 1769.11    2439 1770.71
#Mann= 3 , 0 , 0
       0     .06       0   759.2    .045       0   774.2     .06       0
Bank Sta=759.2,774.2
XS Rating Curve= 0 ,0
Exp/Cntr=0.3,0.1

Type RM Length L Ch R = 1 ,23188   ,454.4,453.4,471.8
XS GIS Cut Line= 3
     1862664.661      301001.391     1862576.456      301535.635
     1862273.604      302757.206
#Sta/Elev= 30
       0 1801.05    19.7 1803.89    78.8 1817.47   118.1  1815.5   226.4 1794.54
   285.5 1767.72   324.9 1759.07   393.8 1733.16   403.6 1732.53   423.3 1725.86
   482.4 1715.93   581.4 1709.55   591.4 1709.31   611.4 1711.16   681.3 1740.43
   691.3 1741.45   781.2 1769.52   791.2 1769.96   841.1 1784.78   851.1  1786.2
     991 1788.73  1220.7 1786.37  1290.6 1784.59  1350.6 1778.29  1380.5 1777.11
  1470.4 1782.13  1570.3 1791.89  1720.1 1789.71  1760.1 1791.78    1800 1796.63
#Mann= 3 , 0 , 0
       0      .1       0   581.4    .045       0   611.4      .1       0
Bank Sta=581.4,611.4
XS Rating Curve= 0 ,0
Exp/Cntr=0.3,0.1

Type RM Length L Ch R = 1 ,22734.1 ,472.3,475.6,478.8
XS GIS Cut Line= 2
      1862162.52      300935.375     1862117.229      302398.849
#Sta/Elev= 30
       0 1791.61    49.8 1803.77    89.6 1809.54   179.3 1806.79   199.2 1801.17
     249 1782.36   268.9 1778.46   338.6  1753.5   358.6 1750.38   438.3 1727.52
   458.2  1723.5   478.1 1714.56   525.5 1709.43   537.9 1709.28   540.5 1709.36
   647.4 1722.82   717.2 1737.86   776.9 1748.36   826.7 1751.45   866.6  1758.4
   886.5  1758.7   966.2 1752.36   986.1  1748.4    1006 1751.56  1035.9 1748.08
  1055.8 1749.27  1115.6 1746.91  1205.2 1746.83  1294.8 1749.62  1464.2 1766.41
#Mann= 3 , 0 , 0
       0      .1       0   525.5    .045       0   540.5      .1       0
Bank Sta=525.5,540.5
XS Rating Curve= 0 ,0
Exp/Cntr=0.3,0.1

Type RM Length L Ch R = 1 ,22258   ,711.9,711.2,708.5
XS GIS Cut Line= 4
     1863541.841      299687.618     1862895.367      300436.751
     1861768.893      301202.531     1861543.857      302460.747
#Sta/Elev= 30
       0 1803.06   139.9 1734.68   199.9 1722.75   289.9 1736.02   389.8 1771.96
   639.7  1812.1   709.6 1801.23   899.6 1735.09   939.5 1738.71  1158.5 1802.57
  1297.7 1791.63  1506.5 1745.08  1645.7 1774.04  1794.8 1791.62  1884.3 1791.45
    2123 1772.33  2272.1 1742.13  2431.5 1729.94  2509.7 1708.91  2524.7 1708.39
  2531.4 1708.24  2631.2 1710.42  2741.1 1731.07    2791 1752.55  2890.9  1775.6
  3180.4 1808.42  3350.2 1807.11  3440.1 1781.54  3569.9  1817.7  3629.8 1841.95
#Mann= 3 , 0 , 0
       0      .1       0  2509.7    .045       0  2524.7      .1       0
Bank Sta=2509.7,2524.7
XS Rating Curve= 0 ,0
Exp/Cntr=0.3,0.1

Type RM Length L Ch R = 1 ,21546.1 ,133.5,134.9,136.3
XS GIS Cut Line= 3
       1862684.5      299540.566     1861335.359      300805.787
     1861286.492      302099.131
#Sta/Elev= 30
       0 1748.02     130  1770.9     190 1787.97   259.9 1791.94   379.9 1787.14
   609.9 1734.56   629.9 1733.77   689.8 1742.09   759.8 1759.77   929.8    1813
  1149.7 1800.08  1349.7 1745.89  1399.7 1738.69  1509.7 1783.52  1589.6 1799.53
  1619.6 1800.19  1749.6 1791.59  1849.6 1774.19  1929.2  1744.6  1969.1 1722.39
  2058.7 1702.76  2062.2 1702.87  2077.2 1703.99    2218 1722.63  2387.2 1768.06
  2546.5 1796.88  2785.4 1803.32  3014.4 1775.62  3064.2 1779.65  3143.8    1799
#Mann= 3 , 0 , 0
       0      .1       0  2062.2    .045       0  2077.2      .1       0
Bank Sta=2062.2,2077.2
XS Rating Curve= 0 ,0
Exp/Cntr=0.3,0.1

Type RM Length L Ch R = 1 ,21410.8 ,514.4,510.6,506.6
XS GIS Cut Line= 2
     1861230.739      300492.898     1861165.953      301717.969
#Sta/Elev= 30
       0 1829.84    59.8 1828.52    99.7 1826.02   129.7 1822.32   179.5 1811.58
   199.5 1808.97   269.3 1787.17   289.2 1783.95   319.2 1773.65     369 1753.33
     389 1748.15   428.9 1725.98   438.8 1721.89   478.7 1717.91   538.6 1704.69
   558.5 1702.81     565 1702.81     580 1703.37   658.3 1713.75   698.2 1717.39
     758 1737.62     768 1738.04   847.8 1764.85   857.8 1767.18   867.7 1767.34
   947.5 1783.58   957.5 1783.64  1037.3 1800.01  1067.2 1802.56  1226.8 1801.91
#Mann= 3 , 0 , 0
       0      .1       0     565    .045       0     580      .1       0
Bank Sta=565,580
XS Rating Curve= 0 ,0
Exp/Cntr=0.3,0.1

Type RM Length L Ch R = 1 ,20900.4 ,434.5,425,414.4
XS GIS Cut Line= 2
     1860743.656      300416.659     1860828.359        301687.2
#Sta/Elev= 30
       0 1800.32    49.7 1792.28    69.6 1790.91   149.2 1777.21   159.2 1776.77
   208.9 1765.71   238.8 1757.33   258.6 1753.78   318.3 1729.71     378 1718.69
   427.8 1705.35   452.5 1703.05   457.6  1702.8   467.5  1702.8   487.5  1703.5
   547.2 1710.98   636.7 1724.31   666.5 1737.09   726.2 1748.72   736.2 1749.56
   825.7 1771.27   855.5 1772.48   895.3 1771.68   925.2  1769.4  1014.7 1751.46
  1044.6 1749.88  1104.2 1764.46  1114.2 1764.34  1163.9 1772.94  1273.4 1781.53
#Mann= 3 , 0 , 0
       0      .1       0   452.5    .045       0   467.5      .1       0
Bank Sta=452.5,467.5
XS Rating Curve= 0 ,0
Exp/Cntr=0.3,0.1

Type RM Length L Ch R = 1 ,20475.5 ,337.8,361.7,386.8
XS GIS Cut Line= 3
      1860389.86      300465.851       1860328.7      300900.263
     1860787.055      301624.287
#Sta/Elev= 30
       0 1821.43    49.8 1811.93   109.7 1809.81   149.6  1804.8   199.4 1792.89
   229.3 1781.72   249.3 1777.66   388.8 1765.25   438.7 1755.35   488.5 1752.98
   558.3 1745.36   677.8 1722.44   744.7 1706.39   759.7 1703.49   767.5 1702.78
   787.4 1704.96   827.3  1719.6   847.2 1722.61   857.2 1722.62   877.1  1717.2
   887.1 1716.47   926.9 1722.61   996.7  1728.9  1016.6 1733.97  1046.5 1744.89
  1066.4 1747.14  1166.1 1775.09  1225.9  1781.7  1275.7  1784.4  1295.6 1783.15
#Mann= 3 , 0 , 0
       0      .1       0   744.7    .045       0   759.7      .1       0
Bank Sta=744.7,759.7
XS Rating Curve= 0 ,0
Exp/Cntr=0.3,0.1

Type RM Length L Ch R = 1 ,20113.7 ,690.1,659.1,627.9
XS GIS Cut Line= 3
     1860324.063      300477.582       1860328.7      301017.543
      1860052.24      301462.284
#Sta/Elev= 30
       0 1804.51      30 1801.14     100 1800.93     150 1795.02     170  1789.1
     180 1788.98     210 1777.15     230 1772.46     260 1769.98     370 1764.38
     450 1749.46     460 1749.31   579.5 1725.21   688.2 1710.26   717.8 1704.18
   735.2 1702.18   737.6 1702.05   750.2 1703.72   777.1 1711.56     787 1712.46
   816.6 1719.66   836.4 1726.88   846.3 1729.34   885.8 1738.38   925.3  1744.5
   945.1  1744.8   984.6 1741.68  1004.4 1741.25  1043.9 1737.23  1063.6 1736.87
#Mann= 3 , 0 , 0
       0      .1       0   735.2    .045       0   750.2      .1       0
Bank Sta=735.2,750.2
XS Rating Curve= 0 ,0
Exp/Cntr=0.3,0.1

Type RM Length L Ch R = 1 ,19454.6 ,418.4,440,461.7
XS GIS Cut Line= 3
     1859488.189      300809.045     1860058.303      301343.323
      1860052.24      301462.284
#Sta/Elev= 30
       0  1759.7    19.8 1763.67    39.6 1768.88    59.3 1775.96   148.4  1780.4
   168.1 1782.51   227.5 1781.14   237.4 1779.32   257.2 1771.35   296.7 1757.68
     356 1737.49   385.7 1728.28   405.5 1720.22     455 1709.61   484.6 1701.16
     493 1699.47   504.4 1698.79     508 1698.99   514.3 1699.33   534.1 1704.73
     544  1706.5   603.3 1709.94   613.2  1711.7   712.1 1738.33   731.9 1744.35
   761.6 1747.83   781.3  1748.7   801.2 1747.54   880.6 1737.96   900.4 1736.87
#Mann= 3 , 0 , 0
       0      .1       0     493    .045       0     508      .1       0
Bank Sta=493,508
XS Rating Curve= 0 ,0
Exp/Cntr=0.3,0.1

Type RM Length L Ch R = 1 ,19014.6 ,633.7,618.6,605.1
XS GIS Cut Line= 3
      1859400.19      300677.965     1859553.345      301069.668
     1859471.553      301665.884
#Sta/Elev= 30
       0 1780.25    29.3 1767.14    39.1 1765.43    68.5 1756.16      88  1753.7
   117.4 1752.64   195.6  1754.5   264.1 1761.62   381.5  1752.8   420.6 1746.22
   440.3 1741.28     460 1740.79   519.2 1725.76   548.8  1720.6   588.3 1716.38
   637.6  1706.6   657.4 1704.28   677.1 1699.56     687 1698.84   688.2 1698.95
   696.8 1699.76   703.2 1702.75   716.6 1710.74   726.4 1715.05   746.1 1718.68
   795.5 1738.75   815.2 1744.58     904 1747.33   992.8 1759.65  1022.4 1758.21
#Mann= 3 , 0 , 0
       0     .06       0   688.2    .045       0   703.2     .06       0
Bank Sta=688.2,703.2
XS Rating Curve= 0 ,0
Exp/Cntr=0.3,0.1

Type RM Length L Ch R = 1 ,18396   ,377.8,385.8,392.2
XS GIS Cut Line= 3
     1858676.871       300804.17     1859099.761      301471.664
     1859909.934      302134.786
#Sta/Elev= 30
       0 1743.22      70 1761.68     190 1781.93   270.1 1783.34   350.1 1768.74
   380.1 1755.87   430.1  1724.7   470.1  1713.5   490.1 1710.89   530.1 1699.06
   537.1 1698.86   540.1 1698.78   552.1 1698.89   590.1 1705.46   630.1 1706.92
   680.2 1714.16   760.2 1734.99   899.9 1732.33  1059.4 1737.51  1109.2 1741.33
    1189 1742.51  1298.7 1741.32  1378.5 1735.67  1418.4 1736.13  1488.2 1732.61
    1558 1735.05  1637.7 1734.76  1697.5 1737.19  1717.5 1741.97  1837.1 1752.51
#Mann= 3 , 0 , 0
       0      .1       0   537.1    .045       0   552.1      .1       0
Bank Sta=537.1,552.1
XS Rating Curve= 0 ,0
Exp/Cntr=0.3,0.1

Type RM Length L Ch R = 1 ,18009.6 ,482.5,497.9,513.3
XS GIS Cut Line= 3
     1858619.448      300839.157     1858830.114      301972.077
     1859006.035      302522.645
#Sta/Elev= 30
       0 1735.07    19.9 1740.02    59.6 1745.61    99.3 1755.04   218.6 1771.23
   258.3 1773.55   347.7  1769.9   397.4 1765.31   427.2  1757.6   437.1 1757.07
   556.3 1732.21   586.1  1725.3   615.9 1715.57   645.7 1709.48   724.5 1701.42
   739.5 1699.05     745 1698.81     755 1699.56   774.8 1708.96   784.8 1711.13
   953.7 1714.91  1102.7 1734.09    1242 1737.74  1281.9 1736.78  1311.8 1735.36
  1401.5 1723.34  1451.3  1720.6  1521.1 1722.75  1590.8 1721.71  1730.3 1729.12
#Mann= 3 , 0 , 0
       0      .1       0   724.5    .045       0   739.5      .1       0
Bank Sta=724.5,739.5
XS Rating Curve= 0 ,0
Exp/Cntr=0.3,0.1

Type RM Length L Ch R = 1 ,17511.4 ,350.2,343,335.9
XS GIS Cut Line= 4
     1858482.068      300827.456     1858465.241      301206.496
     1858164.612      301763.086     1858185.071      302532.418
#Sta/Elev= 30
       0 1754.37   159.8 1725.56   169.7 1725.48   219.7 1737.13   259.6 1742.82
   319.5  1745.6   379.4 1742.57   438.7 1730.25   527.7 1700.48   550.8 1696.72
   557.3 1696.11   565.8 1697.82   596.9  1703.9     755 1712.28   774.8 1726.08
   784.7 1728.96   932.9 1755.76   952.7 1757.59    1112 1762.59  1261.9 1762.22
  1281.9  1760.8  1331.8 1748.17  1381.8 1740.63  1451.8  1740.5  1571.7 1763.04
  1611.7 1775.22  1631.7 1778.53  1691.6 1798.26  1761.6 1799.53  1781.6 1803.84
#Mann= 3 , 0 , 0
       0      .1       0   550.8    .045       0   565.8      .1       0
Bank Sta=550.8,565.8
XS Rating Curve= 0 ,0
Exp/Cntr=0.3,0.1

Type RM Length L Ch R = 1 ,17168.2 ,211,222.6,234.3
XS GIS Cut Line= 3
     1858280.313      300789.933     1858077.563      301206.496
     1857943.526      301876.446
#Sta/Elev= 30
       0 1799.45      69  1786.2    88.7 1784.19   177.4 1761.13   187.3 1761.01
     207 1756.34   256.3 1756.96   285.9 1755.36   325.3 1744.49     345  1742.2
   364.7 1737.45     414 1729.58     493 1709.82   542.5 1703.57   572.2 1701.32
   602.1  1696.4   611.8 1693.08   617.1 1693.83   621.7 1694.48   641.5 1703.54
   700.9 1714.12   720.7 1727.09   740.5 1732.22   760.3 1734.26   879.2 1738.97
     899 1740.77   968.3 1757.39   988.1 1759.54  1047.5 1773.43  1146.5 1784.34
#Mann= 3 , 0 , 0
       0      .1       0   602.1    .045       0   617.1      .1       0
Bank Sta=602.1,617.1
XS Rating Curve= 0 ,0
Exp/Cntr=0.3,0.1

Type RM Length L Ch R = 1 ,16945.3 ,413.6,406.7,399.7
XS GIS Cut Line= 3
     1858208.923      300750.759     1857930.963       301170.66
     1857498.636       301653.52
#Sta/Elev= 30
       0 1799.65    59.2 1792.11   108.6 1779.58     158 1777.08   207.4 1777.08
   246.8 1773.78   276.5 1769.13   325.8    1759   345.6 1752.46   355.5 1751.49
   404.8 1735.99   424.6 1732.14   464.1 1717.38   483.8 1711.99   563.4 1701.46
   592.6 1691.78   593.3 1691.62   607.6 1693.13   643.2 1705.12   673.1 1709.76
     703 1722.05   752.8 1739.56   802.7  1745.3   842.6 1745.33   872.5 1748.61
   922.4 1762.09   942.3 1770.34   982.2    1779    1052 1783.87  1151.7 1800.65
#Mann= 3 , 0 , 0
       0      .1       0   592.6    .045       0   607.6      .1       0
Bank Sta=592.6,607.6
XS Rating Curve= 0 ,0
Exp/Cntr=0.3,0.1

Type RM Length L Ch R = 1 ,16538.6 ,587,560.7,534.4
XS GIS Cut Line= 3
     1857754.148      300582.084     1857546.511      301069.003
     1857347.779      301677.782
#Sta/Elev= 30
       0 1732.37      40 1733.07    59.9 1730.65    69.9 1727.78    99.9 1724.95
   159.8  1728.6   199.8 1727.72   279.6 1715.07   289.6 1715.31   389.5 1700.45
   429.5 1689.55   430.2 1689.55   445.2 1690.94   469.4 1699.74   479.4 1701.77
   499.4 1705.46   529.3 1707.65   549.4 1718.07   559.4 1719.05   579.4 1729.82
   589.4 1733.52   609.4 1736.13   679.4 1751.22   709.4 1751.02   749.5 1747.18
   899.6 1770.06   979.6 1787.08  1029.6 1794.04  1129.7 1803.18  1169.7 1803.48
#Mann= 3 , 0 , 0
       0      .1       0   430.2    .045       0   445.2      .1       0
Bank Sta=430.2,445.2
XS Rating Curve= 0 ,0
Exp/Cntr=0.3,0.1

Type RM Length L Ch R = 1 ,15977.8 ,283.2,289.8,293.2
XS GIS Cut Line= 3
     1856709.374      300595.433     1857227.279       301141.34
     1857275.684       301606.86
#Sta/Elev= 30
       0 1741.46    29.7 1737.35    59.4 1736.09   108.9 1727.38   168.3 1713.69
   188.1 1712.24   247.5 1720.27   287.1 1727.99   306.9 1734.07   336.6 1737.52
   356.4 1737.53   386.2 1733.68     406 1728.99   425.8 1719.21   445.6 1714.37
   485.2 1700.19     505 1691.01   517.1 1688.61   524.8  1688.6   532.1 1689.76
   623.8 1697.87   653.5 1702.48   712.9 1703.86   762.4  1717.1   842.1 1733.62
   901.9 1751.03   921.8 1754.23  1001.4 1776.75    1101 1789.47  1220.5  1798.3
#Mann= 3 , 0 , 0
       0      .1       0   517.1    .045       0   532.1      .1       0
Bank Sta=517.1,532.1
XS Rating Curve= 0 ,0
Exp/Cntr=0.3,0.1

Type RM Length L Ch R = 1 ,15688   ,254.1,260.4,269.9
XS GIS Cut Line= 3
     1856627.106      300649.381     1856907.022      301205.124
      1857210.76      301646.488
#Sta/Elev= 30
       0 1721.51    29.6 1718.59   108.6 1718.44   177.8 1723.83   187.7 1723.12
   246.9 1722.71   266.7 1720.91   355.6 1701.04   375.3 1698.49   434.6 1697.48
   493.8 1692.75   513.6  1692.6   543.2 1690.24   614.8 1687.57   629.8 1687.22
     652 1686.71   661.9  1688.6   681.8  1696.7   691.7 1699.46   701.6 1700.55
   731.4  1700.7   751.2 1705.89   800.8 1728.19   820.7 1738.26   840.5  1744.3
   860.4 1747.66   959.6 1777.25  1009.2 1782.95  1088.6 1790.22    1158  1798.7
#Mann= 3 , 0 , 0
       0      .1       0   614.8    .045       0   629.8      .1       0
Bank Sta=614.8,629.8
XS Rating Curve= 0 ,0
Exp/Cntr=0.3,0.1

Type RM Length L Ch R = 1 ,15426.9 ,625.6,600.2,574.7
XS GIS Cut Line= 3
     1856624.587      300848.138     1856686.485      301473.635
     1857150.864      301678.414
#Sta/Elev= 30
       0 1743.21    49.9 1750.03    59.9  1749.9    89.8 1752.14   109.8 1752.51
   119.7 1751.49   139.7 1744.93   149.7 1744.43   159.6 1741.04   239.4 1709.91
   259.4 1709.07   299.3 1698.19   339.2 1688.96   376.8 1686.44   391.8 1685.34
   409.1  1683.9     419 1684.01     439 1686.57   508.8 1700.23   648.4 1697.51
   668.4 1698.22   718.1 1709.15   728.1 1712.72   797.7 1730.33   817.6 1736.12
   827.6 1741.32   887.3 1760.89   917.1 1768.92  1076.4 1783.65  1136.1 1791.65
#Mann= 3 , 0 , 0
       0      .1       0   376.8    .045       0   391.8      .1       0
Bank Sta=376.8,391.8
XS Rating Curve= 0 ,0
Exp/Cntr=0.3,0.1

Type RM Length L Ch R = 1 ,14826.8 ,300.6,315.4,330.3
XS GIS Cut Line= 2
     1855959.357      301478.676      1857098.34      301801.987
#Sta/Elev= 30
       0    1785    29.8 1789.98   119.4 1798.91   159.2 1801.48   179.1 1799.75
     199 1791.55   268.6 1774.08   278.6 1769.57   348.2 1753.44   447.7  1719.8
   467.6 1715.07   477.6 1711.48   507.4 1693.33   517.4 1690.18   567.1 1685.36
   639.2 1682.35   654.2 1681.61   656.7  1681.5   676.6 1684.43   696.5  1691.9
   716.4 1694.08   766.1 1708.13     786 1715.91   845.7 1731.77   865.6 1739.62
   935.2 1757.95   945.2 1763.46   965.1 1768.64  1094.4 1787.74    1184 1803.84
#Mann= 3 , 0 , 0
       0     .06       0   639.2    .045       0   654.2     .06       0
Bank Sta=639.2,654.2
XS Rating Curve= 0 ,0
Exp/Cntr=0.3,0.1

Type RM Length L Ch R = 1 ,14511.4 ,332,323.3,314.7
XS GIS Cut Line= 3
     1855915.692      301544.318     1856240.167      301659.329
      1856739.58      302334.982
#Sta/Elev= 30
       0 1782.86    29.5 1777.78    98.4 1783.89   216.4 1782.63   275.4 1768.89
   314.8 1762.92   374.3 1748.18   404.3 1737.46   444.3 1720.61   454.3 1719.08
   494.3 1697.27   514.3 1689.55   544.3  1686.2   594.3 1685.95   635.3 1679.94
   644.3 1678.71   650.3 1678.75   664.3 1680.71   694.3 1690.86   734.3 1694.24
   744.4 1696.59   764.4 1706.05   804.4 1721.07   824.4  1725.4   904.4 1757.39
   944.4 1766.33  1034.4 1791.54  1074.4 1792.64  1134.4 1789.78  1184.4 1797.87
#Mann= 3 , 0 , 0
       0     .06       0   635.3    .045       0   650.3     .06       0
Bank Sta=635.3,650.3
XS Rating Curve= 0 ,0
Exp/Cntr=0.3,0.1

Type RM Length L Ch R = 1 ,14188   ,304.9,297.6,290.2
XS GIS Cut Line= 3
     1855704.399      301786.949     1856157.376      302067.344
     1856684.343      302396.182
#Sta/Elev= 30
       0 1807.94    59.2 1801.43    78.9 1802.39   138.1 1800.66   157.8 1797.48
   167.7 1793.68   246.6 1776.72   345.3 1744.03   355.2 1738.16     365 1734.28
   434.1 1710.99   453.8 1702.13   525.2 1678.86   532.7 1677.51   540.2 1678.33
   572.2 1682.92   631.3 1688.11   700.4 1690.94   710.2 1693.55   729.9 1702.96
   749.6  1715.4   759.5 1718.04   828.5  1732.7   848.2 1738.63   917.3 1752.61
     937 1758.91  1015.9 1770.06  1104.6 1787.51  1124.3 1793.12  1153.9 1798.16
#Mann= 3 , 0 , 0
       0     .06       0   525.2    .045       0   540.2     .06       0
Bank Sta=525.2,540.2
XS Rating Curve= 0 ,0
Exp/Cntr=0.3,0.1

Type RM Length L Ch R = 1 ,13890.3 ,316.9,338.9,361
XS GIS Cut Line= 3
     1855583.827      302061.674     1855875.294      302294.599
     1856846.117      302525.903
#Sta/Elev= 30
       0 1747.53    39.3 1746.42   147.3 1753.55   196.4 1752.58   225.8  1754.5
   265.1 1754.72   343.6 1750.48   393.1 1741.45     433 1731.63   452.9 1723.67
   512.8  1706.8   532.8 1699.02   612.6 1678.36   619.7 1677.69   622.6 1677.41
   634.7 1677.66   682.5  1683.9   702.4  1688.4   742.4  1689.3   752.3 1691.03
   782.3 1703.37   832.2 1714.15   852.1  1722.8     902  1736.8  1001.8 1750.91
  1081.7 1765.78  1101.6 1772.12  1211.4 1796.83  1311.2 1803.03  1371.1 1803.27
#Mann= 3 , 0 , 0
       0     .06       0   619.7    .045       0   634.7     .06       0
Bank Sta=619.7,634.7
XS Rating Curve= 0 ,0
Exp/Cntr=0.3,0.1

Type RM Length L Ch R = 1 ,13551.4 ,172.5,177.7,182.9
XS GIS Cut Line= 3
     1855548.277      302128.556     1855914.387      302415.138
     1856184.703      303120.968
#Sta/Elev= 30
       0 1722.99    69.2    1712      89 1710.62   118.7 1720.37   148.4 1725.05
   178.1  1731.8   197.8 1733.64   257.2 1733.55   306.7 1735.38   356.1 1732.69
   395.7 1729.41   445.2 1721.03   544.5 1698.52   564.4 1691.76   584.3  1688.3
   614.1 1678.29   691.9 1674.88   693.7 1674.81   706.9 1678.02   723.5 1684.24
   763.3 1686.64   852.8 1697.58   932.4 1724.25   942.3 1726.62   952.2 1726.73
  1021.9 1744.42  1041.8 1746.14  1061.6 1744.21  1141.2 1753.75  1220.8 1755.73
#Mann= 3 , 0 , 0
       0      .1       0   691.9    .045       0   706.9      .1       0
Bank Sta=691.9,706.9
XS Rating Curve= 0 ,0
Exp/Cntr=0.3,0.1

Type RM Length L Ch R = 1 ,13373.7 ,331.8,315.3,298.6
XS GIS Cut Line= 3
     1855478.636      302160.432     1855787.333      302395.591
     1855898.098      303213.297
#Sta/Elev= 30
       0 1703.41    29.8 1701.74    49.8 1702.59    99.5 1697.91   149.3 1696.67
   169.2 1698.78   189.1 1712.14   218.9 1717.41   288.6 1720.02   358.2 1719.32
   388.1 1721.43   467.6 1706.65   517.3 1701.63     577 1699.62   586.9 1695.43
   616.7 1675.99   626.7 1674.15   636.6 1676.02   666.4  1683.7   726.1  1685.4
   765.8 1690.96   805.6 1698.87   825.5 1703.39   845.4 1711.58   855.3 1713.07
   944.8 1745.05   954.8 1745.97   994.5 1755.93  1103.9 1766.02  1213.2 1771.67
#Mann= 3 , 0 , 0
       0      .1       0   616.7    .045       0   636.6      .1       0
Bank Sta=616.7,636.6
XS Rating Curve= 0 ,0
Exp/Cntr=0.3,0.1

Type RM Length L Ch R = 1 ,13058.3 ,333,348.6,364.3
XS GIS Cut Line= 3
     1855111.737      302349.942     1855738.467       302913.58
     1855885.876      303233.336
#Sta/Elev= 30
       0 1780.91    49.6  1776.5   138.8 1771.76   247.9  1751.1   267.7 1745.09
   317.3 1732.15   327.2 1730.38     357 1722.03   386.7 1710.87   446.2 1692.77
   466.1  1688.8     476 1685.84   495.8 1676.81   505.7 1674.31   515.7 1674.08
   525.6 1674.56   555.3 1679.73     595 1683.89   614.8    1685   684.2 1685.75
   704.1 1687.44   723.9 1694.86   743.7 1700.67   763.6 1704.08     833  1724.7
   852.7 1728.52   999.4 1744.46  1028.7 1750.73  1048.3 1753.77    1195 1765.52
#Mann= 3 , 0 , 0
       0      .1       0   505.7    .045       0   525.6      .1       0
Bank Sta=505.7,525.6
XS Rating Curve= 0 ,0
Exp/Cntr=0.3,0.1

Type RM Length L Ch R = 1 ,12709.8 ,338.2,341.9,345.5
XS GIS Cut Line= 3
     1855058.076      302390.797     1855321.469      302675.761
     1855453.037      303510.157
#Sta/Elev= 30
       0  1791.1   169.2 1781.36     199 1777.51   238.8 1769.84   268.6 1757.92
   318.4 1743.38   368.2 1731.67     388 1724.44   447.7 1714.72   477.5 1711.55
   507.3 1711.06   566.9  1701.9   576.9 1699.24   596.7 1687.85   606.7 1684.56
   646.4 1678.12   699.2 1673.99     706 1673.98   714.2 1674.32   745.8 1684.67
   765.7    1688   835.2 1710.38   855.1 1713.58   934.6 1737.56   954.5 1740.33
  1024.1 1759.15  1063.8 1767.23  1113.5  1774.2  1212.9 1786.15  1232.8 1786.86
#Mann= 3 , 0 , 0
       0      .1       0   699.2    .045       0   714.2      .1       0
Bank Sta=699.2,714.2
XS Rating Curve= 0 ,0
Exp/Cntr=0.3,0.1

Type RM Length L Ch R = 1 ,12367.9 ,274.8,279.9,282.7
XS GIS Cut Line= 3
     1854978.699      302395.635     1855038.041      302613.863
     1855030.458      303500.116
#Sta/Elev= 30
       0 1801.16    39.3 1798.77   108.2  1797.3     118 1795.47   147.5 1786.22
   157.3 1785.71   167.2 1783.26   226.2 1763.46   246.1 1755.64     266 1751.65
   335.7 1723.77   355.6 1719.96   435.3 1692.17   455.2 1689.45     495 1681.16
   561.9 1673.04   574.7 1671.69   576.9 1671.77   584.6 1672.04   614.5 1678.51
   634.4 1680.64   714.1 1695.68     734  1697.6   803.7 1710.33   913.3 1719.21
     983 1718.91  1012.9 1720.25  1092.5 1736.78  1102.5 1736.82  1112.4  1738.7
#Mann= 3 , 0 , 0
       0      .1       0   561.9    .045       0   576.9      .1       0
Bank Sta=561.9,576.9
XS Rating Curve= 0 ,0
Exp/Cntr=0.3,0.1

Type RM Length L Ch R = 1 ,12088   ,293.3,300,309.7
XS GIS Cut Line= 3
     1854890.628      302391.175     1854756.661      302943.717
     1854684.679      303480.937
#Sta/Elev= 30
       0 1803.69    59.8 1801.72    89.8 1797.63   129.7 1786.53   149.6 1779.64
   169.6 1775.88   239.4 1750.61   259.3 1746.76   329.2 1723.83   339.1 1720.99
   349.1 1720.77   438.9 1693.48   448.9 1692.49   498.7 1680.17   561.1 1672.44
   568.6 1671.74   576.1 1672.05   588.3 1674.28   617.8 1682.57   637.5 1685.42
   726.2 1712.52   736.1 1712.64   765.6 1720.75   814.9 1732.17   834.6 1734.26
   903.6 1746.94   923.3 1749.12  1002.2 1763.75  1071.2 1771.12  1110.6 1771.44
#Mann= 3 , 0 , 0
       0      .1       0   561.1    .045       0   576.1      .1       0
Bank Sta=561.1,576.1
XS Rating Curve= 0 ,0
Exp/Cntr=0.3,0.1

Type RM Length L Ch R = 1 ,11788   ,602.9,599.9,596.1
XS GIS Cut Line= 4
     1854773.011      302328.547     1854496.162      302800.337
     1854357.995      303019.559     1854223.592      304340.494
#Sta/Elev= 30
       0 1782.81   109.4  1774.2   149.2  1768.2   258.6 1740.91   318.3 1723.35
   348.1 1712.22   437.6 1691.15   537.1 1671.77   539.5 1671.78   554.5 1673.02
   606.8 1683.02   666.6 1707.42   696.5 1712.33   846.1 1712.75     906 1709.54
  1095.7 1715.42  1175.5 1713.75  1235.4 1718.09  1275.4 1714.83  1425.1 1691.66
    1495 1695.26  1544.9 1705.64  1594.8  1720.5  1614.8 1724.28  1764.5 1731.53
  1854.4 1726.77  1914.3 1716.36  1934.2 1715.44  2044.1 1720.32  2133.9 1720.45
#Mann= 3 , 0 , 0
       0      .1       0   539.5    .045       0   554.5      .1       0
Bank Sta=539.5,554.5
XS Rating Curve= 0 ,0
Exp/Cntr=0.3,0.1

Type RM Length L Ch R = 1 ,11188   ,294.4,300,305.7
XS GIS Cut Line= 4
     1854180.202      302016.302      1853968.07      302519.406
     1853811.362      302896.018      1853708.86      304353.526
#Sta/Elev= 30
       0 1794.06   148.9 1762.92   228.3  1737.1   327.6 1714.43   538.5  1672.2
   553.5  1671.5     556 1671.31   675.3 1697.36   914.1 1726.42   963.9 1729.31
    1074 1726.63  1154.1 1717.16  1234.1 1701.88  1264.2 1700.42  1434.3  1724.5
  1494.3 1729.01  1544.4  1722.9  1614.4 1706.01  1654.4 1702.86  1834.6 1718.81
  1894.6 1727.58  1934.7 1725.09  2004.7 1706.92  2054.8 1698.96  2124.8 1703.79
  2224.9 1716.07  2244.9 1713.96  2274.9 1703.04    2375 1700.32    2415  1703.7
#Mann= 3 , 0 , 0
       0      .1       0   538.5    .045       0   553.5      .1       0
Bank Sta=538.5,553.5
XS Rating Curve= 0 ,0
Exp/Cntr=0.3,0.1

Type RM Length L Ch R = 1 ,10888   ,275.4,274.5,273.5
XS GIS Cut Line= 3
     1854033.159      301944.479     1853704.432      302380.432
     1853375.705      302816.384
#Sta/Elev= 30
       0 1777.34     139 1750.89   158.8 1744.17   228.3 1726.87   248.2 1723.32
     278 1715.24   297.8 1708.03   337.5 1698.36   357.4 1695.57     417  1684.3
   456.6 1679.54   538.5 1671.84     546 1671.26   553.5 1671.92   565.8 1676.46
   585.7  1687.5   595.6 1689.57   615.5 1697.75   625.4 1699.62   655.2 1700.86
   694.9 1695.96   724.7 1694.44     824 1699.94   883.5 1708.26   933.2 1722.49
     963 1721.81  1002.6 1719.26  1032.4 1715.86  1062.2 1714.95    1092 1719.45
#Mann= 3 , 0 , 0
       0      .1       0   538.5    .045       0   553.5      .1       0
Bank Sta=538.5,553.5
XS Rating Curve= 0 ,0
Exp/Cntr=0.3,0.1

Type RM Length L Ch R = 1 ,10613.5 ,673.8,661.7,649.6
XS GIS Cut Line= 4
     1853886.513      301795.679     1853625.543      302023.803
     1853293.687      302501.787     1853214.907      303044.843
#Sta/Elev= 30
       0 1771.84   108.9 1750.11   217.9 1733.96   356.5  1709.8   455.1 1685.53
   474.8 1683.18   537.7 1671.13   543.9 1670.98   552.7 1671.73   593.2 1676.26
   652.4 1699.86     682 1704.66   731.3 1704.55   780.6 1693.38   869.3 1692.05
   908.8 1698.52   998.4 1707.61  1028.3    1706  1098.1 1694.34    1128 1692.53
    1158 1696.09  1207.9 1709.02  1217.8 1709.72  1257.8 1721.89  1267.7 1723.28
  1307.6 1723.62  1367.5 1727.12  1427.4 1727.61  1447.3 1726.23  1477.2 1720.81
#Mann= 3 , 0 , 0
       0      .1       0   537.7    .045       0   552.7      .1       0
Bank Sta=537.7,552.7
XS Rating Curve= 0 ,0
Exp/Cntr=0.3,0.1

Type RM Length L Ch R = 1 ,9951.8  ,596.2,577.7,559.3
XS GIS Cut Line= 3
     1853005.176       301362.87     1852926.989      301721.227
     1852845.544      302952.674
#Sta/Elev= 30
       0 1761.04    79.3 1753.09   128.9 1746.32   178.4 1742.78   257.7 1733.77
   366.8 1729.41   396.6 1724.96   436.5 1716.24   555.9 1705.02   645.5 1686.91
   655.4 1686.91   665.4 1684.87   705.2 1675.99   725.1 1669.34     732 1668.82
     745 1668.56     747 1668.72   774.8 1673.81   844.5 1676.87   864.4 1679.84
   894.3 1686.45   924.1 1696.18   934.1 1696.96   973.9 1712.08   993.8 1717.08
  1212.8  1732.2  1352.1 1737.04  1441.7 1734.08  1521.3 1725.04  1600.9 1710.32
#Mann= 3 , 0 , 0
       0      .1       0     732    .045       0     747      .1       0
Bank Sta=732,747
XS Rating Curve= 0 ,0
Exp/Cntr=0.3,0.1

Type RM Length L Ch R = 1 ,9374    ,620.5,636,651.6
XS GIS Cut Line= 4
     1852342.331      301550.171     1852278.688      301985.109
     1852724.742        302490.3     1852637.046       303017.83
#Sta/Elev= 30
       0 1714.25    99.9 1720.63   149.8 1718.45   229.8 1708.52   379.6 1702.03
   439.6 1702.31   459.4 1698.63     499 1685.28   528.8 1669.08     535  1667.5
   538.7 1666.56     550 1666.74   598.1 1673.14   776.5 1674.19   826.1  1676.4
   855.8 1693.45   885.6 1699.66   974.8  1706.8    1064 1709.75  1113.5 1715.29
  1153.1 1713.27  1192.7  1719.8  1232.3 1728.86  1281.8 1735.83  1390.8  1742.2
  1440.3 1747.59  1509.6 1749.22    1579 1754.27  1588.8 1752.47  1648.3  1732.3
#Mann= 3 , 0 , 0
       0     .06       0     535    .045       0     550     .06       0
Bank Sta=535,550
XS Rating Curve= 0 ,0
Exp/Cntr=0.3,0.1

Type RM Length L Ch R = 1 ,8738    ,460.3,498.8,537.3
XS GIS Cut Line= 3
     1852315.827      301585.997     1852203.759      302226.185
     1852226.563      303161.173
#Sta/Elev= 30
       0 1722.06      50 1725.32      80 1725.33     360 1710.05     380 1709.61
     440 1712.08   489.9 1704.85   529.9 1700.76   589.9 1701.56   649.9  1698.7
   719.6 1697.82   799.2 1691.35   868.8 1677.22     993 1665.95   998.2  1665.7
    1008 1666.53    1028 1672.08  1057.9 1683.24  1077.8 1687.19  1157.4 1718.09
  1177.2 1721.56  1207.1 1730.47  1246.9 1736.49  1306.6 1740.14  1366.3  1741.8
  1455.8 1752.01  1475.7 1755.95  1545.4 1777.02  1555.3 1777.45  1585.2 1788.04
#Mann= 3 , 0 , 0
       0     .06       0     993    .045       0    1008     .06       0
Bank Sta=993,1008
XS Rating Curve= 0 ,0
Exp/Cntr=0.3,0.1

Type RM Length L Ch R = 1 ,8239.2  ,528.2,511.7,495.2
XS GIS Cut Line= 4
     1852240.142      301518.323      1852187.47      302183.834
      1851773.05      302147.438     1851275.287      302578.027
#Sta/Elev= 30
       0 1738.87    69.8 1743.24   139.5 1744.01   428.4 1723.26   468.3 1719.29
   587.9 1699.23   667.6 1695.96   786.4 1669.46   850.2  1664.1   855.8 1664.02
   865.2 1664.61   885.5 1667.91   925.1 1680.48     935 1682.04   984.6 1682.18
  1004.4 1689.37  1014.3 1695.69  1024.2 1704.82    1044 1710.52  1063.8 1713.32
  1103.6 1714.39  1183.3 1720.51  1243.2 1727.84  1263.1 1731.88  1362.8 1758.28
  1382.8 1761.11  1502.4 1799.69  1602.2 1798.32  1691.9 1788.83  1741.8 1778.41
#Mann= 3 , 0 , 0
       0      .1       0   850.2    .045       0   865.2      .1       0
Bank Sta=850.2,865.2
XS Rating Curve= 0 ,0
Exp/Cntr=0.3,0.1

Type RM Length L Ch R = 1 ,7727.5  ,436.5,439.6,442.2
XS GIS Cut Line= 2
     1852186.986      301463.443     1851281.803      302121.936
#Sta/Elev= 30
       0 1754.61      40 1760.56      60 1759.73      90 1754.36   219.9 1736.36
   259.8 1726.72   279.8 1718.89   349.8 1697.23   359.8 1695.33   379.8 1687.48
   429.8    1672   449.7 1669.74   519.7 1668.05   552.6 1664.03   567.6 1662.33
   569.7 1662.27   579.7 1663.78   619.6 1675.64   629.6 1679.82   649.6 1691.92
   669.6 1701.06   679.6 1704.02   709.6 1710.57   809.5 1724.02   849.5 1727.63
   919.5 1736.64   979.4  1739.9  1019.4 1736.53  1099.4 1735.09  1119.4 1733.29
#Mann= 3 , 0 , 0
       0      .1       0   552.6    .045       0   567.6      .1       0
Bank Sta=552.6,567.6
XS Rating Curve= 0 ,0
Exp/Cntr=0.3,0.1

Type RM Length L Ch R = 1 ,7288    ,310.1,299.9,291.3
XS GIS Cut Line= 3
     1852024.674      301142.223     1851545.144      301398.537
     1851059.012      301671.432
#Sta/Elev= 30
       0 1729.15    79.1 1725.19   118.6 1720.41   158.2 1718.77   207.6 1714.97
   247.2 1713.72   326.2  1706.9   415.2 1691.32   474.5 1673.09   504.2 1667.36
     524 1661.71   536.2 1660.28   551.2 1658.85   553.7 1658.66   573.6 1659.56
   613.4 1666.58   623.4 1669.41   643.3 1677.45   663.2 1683.27   693.1 1688.01
   722.9 1690.65   762.8 1700.43   772.7 1704.45   782.7 1707.09   862.3 1726.15
   941.9 1739.75   961.8 1744.95  1041.5 1760.26  1071.4 1763.34  1101.2 1767.86
#Mann= 3 , 0 , 0
       0      .1       0   536.2    .045       0   551.2      .1       0
Bank Sta=536.2,551.2
XS Rating Curve= 0 ,0
Exp/Cntr=0.3,0.1

Type RM Length L Ch R = 1 ,6988    ,305.6,300,293.2
XS GIS Cut Line= 3
     1851665.009      300735.237      1851345.64      301177.433
     1851000.625      301604.506
#Sta/Elev= 30
       0 1736.71   188.4 1718.09   198.4 1719.78   208.3 1719.64   257.9 1714.71
   317.4 1704.13     357 1687.28   406.6 1674.92   515.7 1659.48   535.6 1658.55
     538 1658.61     553 1659.87   595.4 1667.29   605.4 1670.23   645.3 1687.28
   665.2 1691.65   685.2 1700.34   695.2 1703.34   705.2 1703.81   745.1 1700.09
   775.1 1702.59     795 1706.59     815 1714.29     835 1718.49   864.9 1727.99
   894.8 1735.05   914.8 1736.94  1024.6 1754.03  1034.6 1754.16  1094.5 1764.02
#Mann= 3 , 0 , 0
       0      .1       0     538    .045       0     553      .1       0
Bank Sta=538,553
XS Rating Curve= 0 ,0
Exp/Cntr=0.3,0.1

Type RM Length L Ch R = 1 ,6688    ,296.7,300,303.6
XS GIS Cut Line= 3
     1851286.445      300523.379      1851084.87      301030.807
     1850883.685      301538.391
#Sta/Elev= 30
       0 1775.35    39.7 1771.84    69.5 1764.21    79.4 1764.24     139 1746.63
   158.8 1742.62   178.7 1741.42     268 1716.56   287.9 1713.78   367.3 1689.85
   387.2 1687.18   436.8 1674.66   476.5 1666.24   516.2  1664.6   538.5 1658.17
     546 1656.52   553.5 1658.15   565.8 1663.09   575.8 1664.55   605.6 1665.09
   615.5 1666.49   665.1 1681.17     685 1684.48   774.3 1710.54   794.2 1712.65
   873.6  1727.1   923.2 1733.32   943.1 1734.41   992.7 1741.16    1092 1748.69
#Mann= 3 , 0 , 0
       0      .1       0   538.5    .045       0   553.5      .1       0
Bank Sta=538.5,553.5
XS Rating Curve= 0 ,0
Exp/Cntr=0.3,0.1

Type RM Length L Ch R = 1 ,6388    ,292.2,300.8,309
XS GIS Cut Line= 3
     1851078.569      300449.372     1850804.662      300925.852
     1850525.804      301394.526
#Sta/Elev= 30
       0 1752.28      40 1744.32   109.9 1735.27   239.8 1724.94   279.8 1722.85
   309.8 1719.88   369.7 1707.72   379.7 1706.78   409.7 1697.58   469.7 1673.74
   499.6 1664.03   509.6 1661.11   542.1  1656.1   549.6 1655.42   557.1 1656.47
   559.5  1656.8   579.3 1665.26   599.2 1668.99     619 1669.91   628.9 1671.32
   658.7  1676.5   708.2 1686.98   767.7 1705.54   866.9 1720.97   886.7 1725.12
   906.6 1730.73  1015.6 1749.55  1035.5  1752.1  1065.2 1759.85    1095 1765.24
#Mann= 3 , 0 , 0
       0      .1       0   542.1    .045       0   557.1      .1       0
Bank Sta=542.1,557.1
XS Rating Curve= 0 ,0
Exp/Cntr=0.3,0.1

Type RM Length L Ch R = 1 ,6087.2  ,310.3,299,284.3
XS GIS Cut Line= 3
     1851007.494      300395.177     1850402.198        300874.2
     1850282.259      301224.877
#Sta/Elev= 30
       0  1761.1    29.7 1756.14   128.6 1734.52   158.3 1733.12   296.9 1715.37
   316.7 1709.99   376.1 1687.53   415.6 1676.75   425.5 1672.82   465.1 1665.15
   534.4 1660.21   548.7 1657.59   563.7 1654.17     574  1653.3   583.9 1653.49
   593.8 1655.56   633.4 1674.47   653.2 1681.94     673 1687.21   722.4  1693.3
   732.3 1693.15   771.9 1698.91   879.2 1704.77     928 1712.86   947.5 1714.64
   976.7 1722.44  1035.2 1732.08  1054.8 1733.63  1132.8 1747.03  1142.5 1747.46
#Mann= 3 , 0 , 0
       0      .1       0   548.7    .045       0   563.7      .1       0
Bank Sta=548.7,563.7
XS Rating Curve= 0 ,0
Exp/Cntr=0.3,0.1

Type RM Length L Ch R = 1 ,5788    ,257.8,250.8,247.2
XS GIS Cut Line= 3
     1850599.609      300028.792      1850395.51      300507.015
     1850223.503      301178.933
#Sta/Elev= 30
       0 1791.98      40 1782.15      60 1774.21      80 1769.41     120 1756.41
     220 1738.81     260 1726.58     270 1726.04     360 1701.06     380 1698.03
     460 1675.42     480 1672.16     490 1667.58   512.5 1654.16     520 1652.01
   527.5 1652.25   569.5  1659.3   648.8 1659.91   678.5 1663.07     728 1683.87
   767.7 1695.83   787.5 1699.04   797.4 1699.87   827.1 1694.95     837 1695.94
   856.8 1703.07   866.8 1704.17   995.6 1709.44  1074.8 1718.26  1213.5  1737.7
#Mann= 3 , 0 , 0
       0      .1       0   512.5    .045       0   527.5      .1       0
Bank Sta=512.5,527.5
XS Rating Curve= 0 ,0
Exp/Cntr=0.3,0.1

Type RM Length L Ch R = 1 ,5537.2  ,325.6,311,296.4
XS GIS Cut Line= 3
     1850202.989      299920.336     1850131.801      300714.568
     1850145.634      301162.858
#Sta/Elev= 30
       0 1792.11    49.8 1780.63    69.8 1778.76   139.6 1763.33   159.5 1761.51
   189.4 1755.37   249.2 1732.86   259.2 1732.46   338.9 1701.11   348.9 1701.02
   438.6  1665.8   448.6 1665.49   506.5 1651.72   508.4  1651.5   521.5 1652.24
   558.2 1657.65   657.9  1658.7   717.7 1674.32   737.6 1676.52   777.5 1686.43
   857.2 1700.95   887.1 1692.83   897.1 1693.93     907 1699.23     937 1707.29
  1026.6  1709.3  1086.4 1714.18  1156.2 1714.97  1186.1 1717.38  1245.9 1727.82
#Mann= 3 , 0 , 0
       0      .1       0   506.5    .045       0   521.5      .1       0
Bank Sta=506.5,521.5
XS Rating Curve= 0 ,0
Exp/Cntr=0.3,0.1

Type RM Length L Ch R = 1 ,5226.3  ,315.7,323.3,330.6
XS GIS Cut Line= 3
     1849589.083      300066.547     1850027.552      300743.889
     1850074.564      301182.906
#Sta/Elev= 30
       0 1770.77    29.9  1769.6    49.8 1766.93   109.6 1754.24   199.2 1732.28
   219.2 1729.19     259 1718.89   318.8 1697.93   338.7 1693.34   428.3  1658.6
     518 1648.57   526.9  1648.8   541.9 1649.38   697.3 1653.43   737.1 1655.67
   757.1 1660.23     787 1672.35   806.9 1677.61   846.1 1693.25   855.9 1693.62
   875.6 1687.16   895.2 1686.32     905 1687.12   914.8 1690.36   934.4  1700.2
     954 1702.76  1032.5 1705.67  1140.5 1704.25  1199.3    1713  1248.4  1726.3
#Mann= 3 , 0 , 0
       0      .1       0   526.9    .045       0   541.9      .1       0
Bank Sta=526.9,541.9
XS Rating Curve= 0 ,0
Exp/Cntr=0.3,0.1

Type RM Length L Ch R = 1 ,4902.6  ,367.5,380.5,393.8
XS GIS Cut Line= 3
     1849525.068      300095.904     1849779.959      301050.121
     1849999.467      301218.275
#Sta/Elev= 30
       0 1762.78   159.6  1746.2   269.4 1730.85   339.2 1702.89   359.2 1698.76
     439 1669.16   448.9 1666.23   458.9 1665.44   478.9 1657.51   498.8 1652.81
   568.7 1647.62   668.4 1647.41     711 1644.43     726 1644.33   748.2 1644.03
   768.2 1644.18   788.1 1648.05   798.1 1653.41   818.1 1668.53     828  1671.5
     848 1670.26   877.9 1662.01   897.9 1661.12   927.8 1662.72   957.8 1666.62
    1037 1687.62  1066.7 1692.61  1155.6 1701.96  1244.4 1724.01  1264.2 1725.61
#Mann= 3 , 0 , 0
       0      .1       0     711    .045       0     726      .1       0
Bank Sta=711,726
XS Rating Curve= 0 ,0
Exp/Cntr=0.3,0.1

Type RM Length L Ch R = 1 ,4522.4  ,235.5,234.4,238.2
XS GIS Cut Line= 3
      1849451.84      300100.921     1849467.211      300515.843
     1849187.388      301269.583
#Sta/Elev= 30
       0    1755    49.4    1750   128.5 1737.58   138.4  1737.3   227.4 1721.31
   247.2 1719.55   326.2 1698.06   336.1 1697.86     346 1695.44   415.2 1675.62
   435.1 1673.06   524.4 1652.91     574 1647.63   633.6 1647.02   689.2 1639.98
   693.1 1639.81   704.2 1640.33   732.8 1641.18   742.8 1643.29   792.4 1666.53
   822.2  1678.2   861.9  1684.6   911.5 1696.14   931.4 1697.35   961.1 1696.26
   990.9 1707.43  1000.8 1709.69  1050.5 1712.54  1129.9  1720.8  1219.2 1733.53
#Mann= 3 , 0 , 0
       0      .1       0   689.2    .045       0   704.2      .1       0
Bank Sta=689.2,704.2
XS Rating Curve= 0 ,0
Exp/Cntr=0.3,0.1

Type RM Length L Ch R = 1 ,4288    ,308.4,295.9,278.6
XS GIS Cut Line= 3
     1849381.437      300071.297     1849189.964      300631.717
     1848907.487      301113.385
#Sta/Elev= 30
       0 1758.33    59.2 1745.08      79 1743.64   157.9 1730.41   177.7 1728.84
     227 1719.03   256.6 1710.24   276.4  1706.6   335.6 1683.26   365.2 1669.99
   375.1 1669.44   404.7  1661.1     454 1652.16   483.6 1649.34   542.9 1641.19
   584.7 1637.28   592.2 1636.25   599.7  1636.3   612.2 1638.36     662 1656.89
     672 1659.71     682 1660.64   731.8 1676.68   751.8 1680.09   861.4 1683.49
   901.3 1682.41   931.2 1683.92    1001 1689.73  1100.8 1700.32  1150.6 1703.63
#Mann= 3 , 0 , 0
       0      .1       0   584.7    .045       0   599.7      .1       0
Bank Sta=584.7,599.7
XS Rating Curve= 0 ,0
Exp/Cntr=0.3,0.1

Type RM Length L Ch R = 1 ,3992    ,304.1,303.9,305.7
XS GIS Cut Line= 3
     1848829.489      299954.883     1849027.408      300779.724
     1848830.385      301083.423
#Sta/Elev= 30
       0 1746.97    29.9 1740.57    59.9 1730.62    79.8 1727.34   119.8  1717.2
   139.7 1713.33   279.4 1711.39   339.3 1700.81   359.3 1693.78   379.2 1688.53
   419.1 1666.41   459.1 1642.58     469 1637.85     479 1636.38     489 1633.46
     499 1634.19   518.9 1637.98   548.9 1640.06   628.7 1637.66   678.6 1639.99
   708.5 1644.22   758.4 1655.44   778.4 1657.99   848.2 1670.73   887.4 1671.37
   975.4 1677.64  1063.5 1689.54  1102.6  1691.9  1190.7 1700.68  1210.3 1701.24
#Mann= 3 , 0 , 0
       0      .1       0     479    .045       0     499      .1       0
Bank Sta=479,499
XS Rating Curve= 0 ,0
Exp/Cntr=0.3,0.1

Type RM Length L Ch R = 1 ,3688    ,307.6,316.6,323.7
XS GIS Cut Line= 3
     1848529.417       300023.84     1848662.302      300554.795
     1848746.596      301094.531
#Sta/Elev= 30
       0 1755.28    19.9 1752.02    49.8 1745.13    69.7 1742.85    89.6 1742.38
   139.3 1732.95   179.1 1721.94   189.1 1722.08   278.6 1699.03   298.5 1696.62
   368.2 1678.76   388.1  1675.9   447.8 1656.05   477.7 1642.57   487.6 1641.91
   507.5 1631.88   517.5 1631.28   527.4 1632.32   547.3 1633.84   616.9 1633.81
   696.3 1636.64   706.2 1638.89   765.8 1658.75   795.6  1664.9   875.1 1676.68
     885 1676.85   924.8 1681.64   974.4 1685.09  1063.8 1696.83  1093.6 1699.54
#Mann= 3 , 0 , 0
       0      .1       0   507.5    .045       0   527.4      .1       0
Bank Sta=507.5,527.4
XS Rating Curve= 0 ,0
Exp/Cntr=0.3,0.1
